--- KIAHCR.prj (project) ---

Proj Title=KIAHCR
Current Plan=p01
Default Exp/Contr=0,0
English Units
Geom File=g01
Flow File=f01
Plan File=p01
BEGIN DESCRIPTION:
END DESCRIPTION:
DSS Export Rating Curves= 0
DSS Export Rating Curve Sorted= 0
DSS Export Volume Flow Curves= 0
DXF OffsetX= 0
DXF OffsetY= 0
DXF ScaleX= 0
DXF ScaleY= 0

--- KIAHCR.p01 (plan) ---

Plan Title=Floodplain
Program Version=4.00
Geom File=g01
Flow File=f01
K Sum by GR=0
Std Step Tol=0.01
Critical Tol=0.01
Num of Std Step Trials=20
Max Error Tol=0.3
Flow Tol Ratio=0.001
Split Flow NTrial=30
Split Flow Tol=0.02
Split Flow Ratio=0.02
Log Output Level=0
Friction Slope Method=1
Unsteady Friction Slope Method=2
Unsteady Bridges Friction Slope Method=1
Global Log Level=0
CheckData=False
Run HTab=0
Run UNet=0
Run PostProcess=0
UNET Theta=0
UNET Theta Warmup=0
UNET ZTol=0
UNET ZSATol=0
UNET MxIter=0
UNET MaxInSteps=0
UNET DtIC=0
UNET DtMin=0
UNET MaxCRTS=0
UNET WFStab=0
UNET SFStab=0
UNET WFX=0
UNET SFX=0
UNET DSS MLevel=0
UNET DZMax Abort=0
UNET Convert EG Bridges=0
UNET Use Existing IB Tables=0
UNET Froude Limit=0
UNET Froude Power=0
Write IC File=0
Echo Input=False
Echo Output=False
Write Detailed=0

--- KIAHCR.f01 (steady flow) ---

Flow Title=NFF Regression Equation
Program Version=4.00
Number of Profiles= 1
Profile Names=P100yr
River Rch & RM=KIAHCR,Main            ,48378.8
    1466
River Rch & RM=KIAHCR,Main            ,47949.4
    2108
River Rch & RM=KIAHCR,Main            ,44041.1
    2149
River Rch & RM=KIAHCR,Main            ,43731.2
    2456
River Rch & RM=KIAHCR,Main            ,38934.8
    2543
River Rch & RM=KIAHCR,Main            ,35256
    2821
River Rch & RM=KIAHCR,Main            ,22176.8
    3127
River Rch & RM=KIAHCR,Main            ,21829.3
    3692
River Rch & RM=KIAHCR,Main            ,14929.9
    3871
River Rch & RM=KIAHCR,Main            ,14078.9
    4309
Boundary for River Rch & Prof#=KIAHCR,Main            , 1
Up Type= 0
Dn Type= 3
Dn Slope=0.0002
DSS Import GetInterval= 0
DSS Import GetPeak= 0
DSS Import FillOption= 0

--- KIAHCR.g01 (geometry) ---

Geom Title=USGS 10m DEM
Program Version=4.00

River Reach=KIAHCR          ,Main
Reach XY= 30
     1612950.279       368575.15     1613175.167      369161.885
     1612143.232      370539.257     1612777.647      371264.116
     1612445.971      371979.099     1611286.239      373138.276
     1610868.937      372502.059     1610597.583       373059.04
     1608766.067       372760.22     1608502.946      373413.855
     1608956.531      374275.631     1607805.982      373919.303
     1608363.789      374814.317     1606716.337      376277.345
      1606974.62      377551.964     1606258.283       378660.19
      1607229.08      381021.468     1606562.492      380960.598
     1606338.263      381774.981     1607947.972      383674.456
     1605636.889      384931.645     1605515.705      387219.521
      1604059.28       388976.71     1602210.201      389501.902
     1599209.683      390015.237     1597592.888      389323.007
     1595720.518      389455.067     1596057.388      390755.357
     1594502.807       390777.64     1594403.098      392360.665

Type RM Length L Ch R = 1 ,48378.8 ,117.9,117.8,117.7
XS GIS Cut Line= 4
     1611129.124       368318.47     1612861.349      368704.046
     1613161.919      368322.238      1614005.02      366964.348
#Sta/Elev= 30
    10.1 1111.55    50.7  1129.1   233.2  1189.5   334.6 1193.45   395.5 1187.12
   557.7 1139.62   638.9 1097.76   699.7 1073.26   851.8 1036.25  1024.2  971.93
    1227     912  1287.9  909.22  1531.2   925.1  1774.6  841.13  1921.6   774.1
  1936.6  772.44  1951.6  774.47  2118.8  780.87  2209.9  789.26  2341.5  828.72
  2584.3   875.2  3069.8 1022.73  3100.2 1035.33    3171  1076.7  3191.2 1084.01
  3454.2 1132.64  3514.9 1136.67  3636.3 1126.93  3788.1 1064.86  3858.9  1039.8
#Mann= 3 , 0 , 0
       0      .1       0  1921.6    .045       0  1951.6      .1       0
Bank Sta=1921.6,1951.6
XS Rating Curve= 0 ,0
Exp/Cntr=0.3,0.1

Type RM Length L Ch R = 1 ,48261   ,294.3,311.7,329
XS GIS Cut Line= 4
     1611619.008       368896.56     1612955.152       368776.58
     1613282.371      368356.649     1613773.199      367631.313
#Sta/Elev= 30
    10.2 1201.72   101.6 1183.39   315.1 1128.33   457.3 1070.58   538.6 1045.72
   548.8 1044.25   599.6 1048.72   630.1 1048.11   691.1 1034.77   802.9 1021.42
     996   985.2  1067.1  953.63  1209.4  880.51  1250.1  864.81  1361.6  831.68
  1487.2  773.71  1502.2  772.06  1517.2  774.34  1873.9   784.2    1894  786.93
  1984.6  809.66    2045  816.66  2125.6  833.73  2206.1  862.43  2256.4  885.12
  2387.3  935.03  2628.9  989.24    2649 1000.14  2709.4  1045.9  2749.7  1069.3
#Mann= 3 , 0 , 0
    10.2      .1       0  1487.2    .045       0  1517.2      .1       0
#XS Ineff= 2 , 0
                          1655.1          848.36
Permanent Ineff=
       F       F
Bank Sta=1487.2,1517.2
XS Rating Curve= 0 ,0
Exp/Cntr=0.3,0.1

Type RM Length L Ch R = 1 ,47949.4 ,393,419.2,446.7
XS GIS Cut Line= 4
     1612567.943      368918.375     1613080.586      368945.643
     1613467.795      368814.755     1614417.705      369775.763
#Sta/Elev= 30
    10.1 1012.94    50.3  985.52   100.7  955.08   261.7  882.46     312  862.23
   352.3   848.2   412.7  836.93   523.3  807.42   593.1  780.46   657.9  771.71
   672.9  770.61   687.9  771.31   762.6  777.34   772.6   780.5   852.3  825.06
   922.1  849.77   993.2  871.15  1023.7  883.24  1094.8   917.7  1125.3  928.37
  1440.2  963.42    1613   977.7    1806 1032.09  1907.6 1055.66  2039.7 1093.93
  2070.2 1095.07  2131.1 1090.03  2192.1 1095.15  2232.7 1103.39  2273.3 1120.49
#Mann= 3 , 0 , 0
       0      .1       0   657.9    .045       0   687.9      .1       0
Bank Sta=657.9,687.9
XS Rating Curve= 0 ,0
Exp/Cntr=0.3,0.1

Type RM Length L Ch R = 1 ,47530.2 ,755,751.5,746.2
XS GIS Cut Line= 3
     1612720.645      369054.716       1613102.4      369283.769
      1613445.98      369518.276
#Sta/Elev= 30
    10.1  915.31    40.5  902.68    50.6   897.7   101.2  870.51   131.5  857.36
   141.7  853.62   151.8  850.63   202.4  839.49   232.7  831.21     253  824.28
   323.8   798.2   374.4  780.51   384.5     778   420.1  770.52     425  769.52
   435.1  768.47   445.2  768.94   450.1   770.1   495.9  783.24   546.7  796.15
   556.8  797.92     567  798.86   617.7  799.81   627.8  800.55   648.1  804.22
   678.6  811.36   739.4   831.9   820.6  860.35   840.9  868.12   861.2  877.01
#Mann= 3 , 0 , 0
       0      .1       0   420.1    .045       0   450.1      .1       0
Bank Sta=420.1,450.1
XS Rating Curve= 0 ,0
Exp/Cntr=0.3,0.1

Type RM Length L Ch R = 1 ,46778.7 ,749.9,763.1,776.7
XS GIS Cut Line= 3
     1612387.972      369758.237     1612814.412      369946.719
     1613178.751      370101.816
#Sta/Elev= 30
    10.1  927.29    50.7  912.49    81.1  902.46   101.4  895.01   131.8  881.79
   172.3  860.99   212.8  841.39   304.1  808.57   334.5  796.53   364.9  782.39
     375  778.28   385.2  775.49   395.3  773.99   451.2   768.7   466.2  767.86
   481.2   768.8   486.5  769.53   496.7  772.48   506.9  777.13     517   783.3
   537.3  799.24   547.5   806.6   557.6  812.34   577.9  821.44   618.5  842.05
     649  856.48   720.1  888.24   760.7  907.19   811.4   933.7   862.2  958.98
#Mann= 3 , 0 , 0
       0      .1       0   451.2    .045       0   481.2      .1       0
Bank Sta=451.2,481.2
XS Rating Curve= 0 ,0
Exp/Cntr=0.3,0.1

Type RM Length L Ch R = 1 ,46015.6 ,888.6,836.9,785.2
XS GIS Cut Line= 3
     1611990.798      370100.714     1612371.611      370543.562
     1612524.314       370690.81
#Sta/Elev= 30
    10.1  840.17   130.9  816.38   211.5  801.67   251.8  792.87     292  783.64
   302.1  781.76   312.2  780.34   352.5  777.39   372.6  775.41   382.7  773.95
   392.7  771.46   402.8  768.31   407.9  767.22   412.9  766.15   422.9  765.94
   437.9  767.22   463.2  769.94   473.3  771.49   483.4  774.72   503.5  783.23
   523.6  790.41   604.3  816.46   624.5  822.53   634.6  825.07   644.7  826.68
     675  829.11   715.4  833.75   735.6  835.69     776  838.29   796.2  838.68
#Mann= 3 , 0 , 0
       0      .1       0   407.9    .045       0   437.9      .1       0
Bank Sta=407.9,437.9
XS Rating Curve= 0 ,0
Exp/Cntr=0.3,0.1

Type RM Length L Ch R = 1 ,45178.7 ,752.4,792.6,835.1
XS GIS Cut Line= 3
     1612224.363      371356.156     1612553.989      371021.606
     1612873.347      370696.264
#Sta/Elev= 30
      10  881.37      50  896.23      60  896.89    69.9  894.89   139.9  869.96
   219.8   839.8   269.8  819.64   289.8  809.13   309.8  799.85   369.7  777.65
   389.7  770.95   399.7   768.4   434.7  764.41   449.7  763.28   459.7  764.04
   464.7  765.32   469.7  766.61   520.3  788.68   530.4  792.43   550.7  797.95
   560.8  801.81   601.4  820.43   641.9  841.48   753.3  910.08   763.5  915.82
   773.6  920.74   814.1  936.12   895.2  968.96   905.3   973.5   925.5  984.89
#Mann= 3 , 0 , 0
       0      .1       0   434.7    .045       0   464.7      .1       0
Bank Sta=434.7,464.7
XS Rating Curve= 0 ,0
Exp/Cntr=0.3,0.1

Type RM Length L Ch R = 1 ,44386   ,335.9,344.9,351.8
XS GIS Cut Line= 4
     1612251.631      371448.868      1612648.64      371687.832
     1612843.713      371825.353      1614369.01      372291.627
#Sta/Elev= 30
    10.1  874.89    30.2  877.09    40.3  874.07   221.6  802.15   292.1  771.32
   312.3  768.91     413  769.55   448.4  762.22   463.4  760.74   478.4  765.58
   503.2  775.58   592.7  788.28   672.2  785.23   844.3  784.93   905.2  793.98
  1118.6  796.15  1179.5   808.3  1250.6  811.79  1281.1  819.19  1423.3  873.39
  1484.3  892.36  1545.3  907.37  1596.1  930.58  1636.7  935.44  1738.3  966.42
  1768.8   971.4  1900.8 1014.88  1941.5 1022.85  1982.1 1027.07    2297 1049.95
#Mann= 3 , 0 , 0
       0      .1       0   448.4    .045       0   478.4      .1       0
Bank Sta=448.4,478.4
XS Rating Curve= 0 ,0
Exp/Cntr=0.3,0.1

Type RM Length L Ch R = 1 ,44041.1 ,299.8,309.9,320
XS GIS Cut Line= 4
     1611872.262      371311.674     1612264.243      371763.305
     1612579.532      372112.679     1612945.949       374174.84
#Sta/Elev= 30
    10.1  910.39    81.1  886.84   243.3  823.26   293.9   808.6   324.3     806
   476.4   822.3   527.1  815.71     608  797.72   698.1  765.65   863.4  759.77
   878.4  759.39   893.4  764.24   908.4  771.08   938.5  774.82  1008.5  799.47
  1068.6  795.58  1129.3  803.27  1240.6  809.82  1372.2  824.57  1645.4  847.45
  1797.1  875.58  1999.5  918.77  2100.7  936.46    2303  984.44  2424.5  992.66
  2566.1 1014.11  2707.8 1050.19  2839.3  1059.6  3082.1 1089.78  3163.1 1092.93
#Mann= 3 , 0 , 0
    10.1      .1       0   863.4    .045       0   893.4      .1       0
#XS Ineff= 2 , 0
          773.91  816.78
Permanent Ineff=
       F       F
Bank Sta=863.4,893.4
XS Rating Curve= 0 ,0
Exp/Cntr=0.3,0.1

Type RM Length L Ch R = 1 ,43731.2 ,971.3,960.7,950
XS GIS Cut Line= 4
      1611216.12      370970.821     1612034.167      371746.262
     1612238.679      372240.499     1612562.489      373612.432
#Sta/Elev= 30
    10.2 1131.07   111.7 1141.51   172.6 1140.65   203.1 1134.04   304.6  1097.4
   497.6 1019.87   700.7  933.27   792.1  886.11     853  869.93  1056.1  803.36
  1207.9  780.43  1379.5  763.17  1495.7  761.35  1510.7  758.83  1525.7  761.12
  1561.1  778.41  1601.5  785.64  1702.6  838.69  1885.2  869.35  2118.4  945.25
  2219.8  986.11  2270.5  979.84  2341.5   979.7  2392.2   990.5  2432.8   991.7
  2584.9 1049.14  2605.2 1053.25  2696.5 1054.36  2909.4 1073.02  3071.7 1074.68
#Mann= 3 , 0 , 0
       0      .1       0  1495.7    .045       0  1525.7      .1       0
Bank Sta=1495.7,1525.7
XS Rating Curve= 0 ,0
Exp/Cntr=0.3,0.1

Type RM Length L Ch R = 1 ,42770.5 ,419.4,428.5,437.4
XS GIS Cut Line= 4
     1611396.655      372202.642     1611471.759      372581.352
      1611795.57      372930.726     1612434.669      373586.868
#Sta/Elev= 30
    10.2  921.01    91.4  915.36     193  903.83   274.3  886.13     315  874.49
   345.4  862.16   477.3  793.26   538.1  765.27   558.4  762.08   675.1  758.53
   690.1   756.2   705.1  758.06     751  771.27   761.1  780.26   781.4  805.98
   791.5  815.66   932.9  889.99     953  897.45  1023.5  910.17  1053.7  918.57
    1104  946.31  1124.1  954.36  1204.7   971.4  1265.1   963.9  1325.5  967.21
  1496.6  994.06  1526.8  995.89  1597.2 1013.15  1697.9 1018.28  1778.4  1033.2
#Mann= 3 , 0 , 0
       0      .1       0   675.1    .045       0   705.1      .1       0
Bank Sta=675.1,705.1
XS Rating Curve= 0 ,0
Exp/Cntr=0.3,0.1

Type RM Length L Ch R = 1 ,42342   ,85.4,86.3,87.4
XS GIS Cut Line= 4
     1611368.032      371775.811     1611282.067      372911.776
     1611521.541      373403.005      1612012.77      373943.356
#Sta/Elev= 30
    10.1  986.22    50.4  981.71     121  969.68   272.2  930.02   332.7  919.07
   423.4   898.9   504.1  885.29   655.3  856.08   887.2  818.57  1038.4  789.01
    1109  785.75  1169.6  780.72  1220.2  769.14  1301.1  766.64  1311.3  765.56
  1336.7  757.78  1351.7  756.05  1366.7  758.37  1392.2  763.86  1412.5  770.92
  1442.8  776.78  1564.3  783.96  1726.3  800.39  1807.4  806.86  1898.7  812.03
  2040.7  816.33    2132  830.23  2182.7  833.15  2284.1  858.56    2416  887.82
#Mann= 3 , 0 , 0
       0      .1       0  1336.7    .045       0  1366.7      .1       0
Bank Sta=1336.7,1366.7
XS Rating Curve= 0 ,0
Exp/Cntr=0.3,0.1

Type RM Length L Ch R = 1 ,42255.7 ,904.1,909.9,915.7
XS GIS Cut Line= 4
     1611341.899      371710.325     1611195.707      372911.161
     1611419.707      373414.179     1611324.856      374454.192
#Sta/Elev= 30
    10.1  982.14    90.7  975.02   181.5  958.38   383.1  903.79   433.5  882.99
   473.8  870.42   594.8  845.02   816.5  814.19  1048.4  791.87  1129.1  787.15
  1209.7  773.22  1249.7  775.21  1349.9  772.46  1409.9  767.56    1435  759.79
    1450   755.6    1465  757.19  1540.1  780.41  1630.2  785.65  1710.3  812.66
  1760.3  831.72  2003.7  947.24  2135.5  991.95  2206.5  995.08  2368.7 1035.03
    2389 1033.12  2480.2  1008.6  2530.9 1004.24  2723.6 1050.86  2804.7 1056.59
#Mann= 3 , 0 , 0
       0      .1       0    1435    .045       0    1465      .1       0
Bank Sta=1435,1465
XS Rating Curve= 0 ,0
Exp/Cntr=0.3,0.1

Type RM Length L Ch R = 1 ,41345.8 ,959.2,959.8,957.9
XS GIS Cut Line= 4
     1610909.352      370595.883     1610653.712      371592.878
     1611020.129      373331.229      1611028.65      374634.992
#Sta/Elev= 30
    10.1 1143.94    60.5 1136.93   211.9 1078.76     333 1013.28   393.5  988.01
   474.3  964.68   544.9   962.8   585.3   932.7   645.8  907.97   968.7  844.54
  1069.9  816.05  1191.7   795.7  1293.2  802.69    1415  780.13  1831.2  754.93
  1938.1  754.42  1953.1  754.36  1968.1  754.51  2186.5  756.91  2298.2  768.39
  2409.9  768.42  2460.6  808.13  2805.8   884.2  2997.8  964.94  3139.3   994.4
  3331.4 1065.98  3654.8 1052.31  3897.3 1011.63  4048.9  1047.8  4109.6  1069.4
#Mann= 3 , 0 , 0
       0      .1       0  1938.1    .045       0  1968.1      .1       0
Bank Sta=1938.1,1968.1
XS Rating Curve= 0 ,0
Exp/Cntr=0.3,0.1

Type RM Length L Ch R = 1 ,40386   ,561.1,571.2,580
XS GIS Cut Line= 3
     1610202.082      372189.371     1610351.209      373083.519
     1610415.115       373595.39
#Sta/Elev= 30
    10.1  955.96    90.6  958.75   211.5  956.29   231.7  953.81   271.9  944.15
   292.1     943   352.5  943.22   402.9  954.65     413  954.17   483.5  928.22
   543.9  899.19   594.3  882.55   614.4  874.01   654.7  852.11   715.1   810.9
   805.8  763.61   846.1  755.34   891.5  750.74   906.5  749.84   921.5  752.64
   957.1  763.85   977.3  766.51   997.5  774.44  1230.2  894.02  1260.5  911.32
  1311.1  943.76  1331.3  954.31  1371.8  958.88  1402.1  975.78  1422.3  979.46
#Mann= 3 , 0 , 0
       0      .1       0   891.5    .045       0   921.5      .1       0
Bank Sta=891.5,921.5
XS Rating Curve= 0 ,0
Exp/Cntr=0.3,0.1

Type RM Length L Ch R = 1 ,39814.8 ,878.3,880,881.7
XS GIS Cut Line= 4
     1609810.101      372129.722     1609827.143      372862.556
     1609758.973      373263.058     1610057.219      374072.584
#Sta/Elev= 30
      10  1036.4    90.4 1035.06   291.2  966.73   381.6  957.86   532.2  881.21
   672.8   820.7   773.7  787.23   824.4  777.23   895.5  757.69   951.6  748.26
   966.6  746.88   981.6  748.52    1058  759.76  1139.3  813.85  1200.2  845.98
  1230.6  857.69  1281.4  868.92  1362.6  878.88  1484.4  898.93  1565.6  907.21
  1606.2  916.05  1646.8  928.99  1707.7   938.6    1728  944.49  1768.6  964.34
  1829.5   976.2  1880.2 1002.89  1910.7 1014.09  1971.6 1029.65    2002 1032.15
#Mann= 3 , 0 , 0
       0      .1       0   951.6    .045       0   981.6      .1       0
Bank Sta=951.6,981.6
XS Rating Curve= 0 ,0
Exp/Cntr=0.3,0.1

Type RM Length L Ch R = 1 ,38934.8 ,610.8,572.8,534.8
XS GIS Cut Line= 4
     1608932.404       371286.11     1609060.224      372538.745
     1608975.011      372913.684     1609571.504      373680.603
#Sta/Elev= 30
    10.2 1136.76    50.8 1133.95    71.1 1129.49   345.2 1049.29   629.6 1044.52
   751.4 1031.63   822.5 1006.63   893.6  973.97   934.2  968.82  1005.3  945.47
  1045.9   929.9  1157.6  877.16  1269.3  840.97  1400.8  762.32  1446.5  746.53
  1461.5  745.56  1476.5  747.15  1542.5  763.69  1603.2  763.26  1643.6  778.25
    1755   810.1  1815.7  823.23  1896.7  835.44  1997.9  870.05  2088.9  882.84
  2190.2  889.68  2230.6  895.66  2281.2  894.94  2422.9  884.75  2615.2  862.89
#Mann= 3 , 0 , 0
       0      .1       0  1446.5    .045       0  1476.5      .1       0
Bank Sta=1446.5,1476.5
XS Rating Curve= 0 ,0
Exp/Cntr=0.3,0.1

Type RM Length L Ch R = 1 ,38362   ,1620.5,1626.3,1631.9
XS GIS Cut Line= 4
     1608208.091      372001.902     1608412.603      372905.162
     1608787.541      373126.717     1609963.485      374507.172
#Sta/Elev= 30
    10.1 1012.05    70.5 1025.83   140.9 1022.69   422.8  966.29   664.4  960.05
   704.7  954.24   805.3  919.61   926.1  869.52  1113.7  750.55 1129.38  745.38
  1143.7  750.15  1189.5  763.84  1341.4  760.66  1351.5  766.34  1371.8  796.17
    1392  812.57  1523.7  866.47  1604.8  869.02  1908.7   851.9  1989.7  857.06
  2182.2  892.74  2344.3   936.2  2435.5  936.69  2486.2  918.93  2496.3  919.74
  2567.2  959.71  2648.2  962.56  2779.9 1006.82  2931.9 1049.67  3175.1    1066
#Mann= 3 , 0 , 0
    10.1      .1       0  1113.7    .045       0  1143.7      .1       0
Bank Sta=1113.7,1143.7
XS Rating Curve= 0 ,0
Exp/Cntr=0.3,0.1

Type RM Length L Ch R = 1 ,36735.7 ,1481.7,1479.7,1477.8
XS GIS Cut Line= 4
     1608097.314      372138.243     1608506.338      373774.337
     1609477.769      374583.864     1609954.963      374992.887
#Sta/Elev= 30
    10.2  975.61   132.1  995.04   264.1   964.6   579.1  966.86   721.3  959.52
   751.8  952.68   863.5  910.82   944.8  889.74  1026.1   860.6  1107.4  838.07
    1341  800.07  1412.1   801.1  1534.1  818.78    1656  856.17  1878.7  853.31
    2000  845.92  2070.9   828.4  2202.4  770.22  2298.6  744.41  2313.6  742.92
  2328.6  744.58  2414.8     754  2576.7  835.71  2728.4  922.09  2789.1   942.3
  2839.7  948.03  2991.5 1008.25  3346.3 1057.03  3447.7 1061.48  3579.5 1058.73
#Mann= 3 , 0 , 0
       0      .1       0  2298.6    .045       0  2328.6      .1       0
Bank Sta=2298.6,2328.6
XS Rating Curve= 0 ,0
Exp/Cntr=0.3,0.1

Type RM Length L Ch R = 1 ,35256   ,912.3,876.1,839.8
XS GIS Cut Line= 4
     1606682.774      373510.176     1607500.821      373680.603
     1608208.091      374225.968     1609366.992      374992.887
#Sta/Elev= 30
    10.1 1101.62   100.7 1120.93   140.9  1118.5   362.4 1031.77   553.7  998.28
   815.5  944.77   876.2  944.49   947.3  910.81  1018.3  864.11  1150.2  752.21
  1170.5  744.98  1206.3   742.7  1221.3  741.19  1236.3  741.72  1464.9  744.83
  1505.4   749.4  1647.5  784.54  1759.2     797  1880.9  820.16  2063.5  849.15
    2175  851.38  2266.3  860.43  2317.1  872.13  2499.6  924.24  2540.2   931.9
  2601.1  933.19  2641.7  941.24  2722.8  968.33  2854.7  1002.8  3118.4 1012.37
#Mann= 3 , 0 , 0
       0      .1       0  1206.3    .045       0  1236.3      .1       0
Bank Sta=1206.3,1236.3
XS Rating Curve= 0 ,0
Exp/Cntr=0.3,0.1

Type RM Length L Ch R = 1 ,34379.9 ,408.5,440.4,472.4
XS GIS Cut Line= 4
     1606998.063      374277.096     1608037.665      374720.205
     1608463.731      374464.565     1609401.077      375146.271
#Sta/Elev= 30
    10.1 1137.38    80.7 1123.64   232.1 1104.62   343.1 1079.29   484.3 1016.47
     565  987.64   635.7  980.88   867.8  930.02   928.3  924.47  1049.4  885.32
  1130.1  851.13  1201.1  831.51  1241.6  809.31  1282.2  779.24    1343   751.9
  1363.3  745.68  1429.4   740.2  1444.4  739.49  1459.4  740.73  1495.1  749.84
    1627  824.58  1788.2  860.44  1909.2  906.95  1999.9  935.05  2060.3  929.29
  2100.7  932.62  2191.4  960.81  2292.2 1000.37  2503.8 1000.93    2786  991.38
#Mann= 3 , 0 , 0
       0      .1       0  1429.4    .045       0  1459.4      .1       0
Bank Sta=1429.4,1459.4
XS Rating Curve= 0 ,0
Exp/Cntr=0.3,0.1

Type RM Length L Ch R = 1 ,33939.5 ,197,199.5,202
XS GIS Cut Line= 4
     1607331.118       374485.19     1608146.557      374878.172
     1608426.557      375040.278      1609227.26      375595.366
#Sta/Elev= 30
    10.1 1078.85    60.3 1059.98   140.8 1025.13     171 1015.45   372.1  983.02
   452.6  962.21   563.2  928.67   583.3  928.18   603.5  923.08   633.6  911.96
   683.9   888.9   945.6  754.59   965.9  748.98  1041.9   739.8  1056.9  738.29
  1071.9  738.48  1097.3   740.7  1117.5  745.43  1188.3  779.95  1208.5  785.78
  1279.5  789.77  1411.4  792.83  1665.1  807.54  1837.7   806.9  1888.4  812.29
  1918.9  813.04  1989.9     833  2101.5  871.54  2142.1  880.48    2203   903.1
#Mann= 3 , 0 , 0
       0      .1       0  1041.9    .045       0  1071.9      .1       0
Bank Sta=1041.9,1071.9
XS Rating Curve= 0 ,0
Exp/Cntr=0.3,0.1

Type RM Length L Ch R = 1 ,33740   ,368.1,379,388.7
XS GIS Cut Line= 4
     1607298.615      374602.209     1608014.407      375002.712
     1608414.909      375283.916     1609181.828       375888.93
#Sta/Elev= 30
    10.1 1085.88   101.3 1081.29   192.4 1061.61   222.8 1050.87   273.4 1025.99
   394.9  995.26   577.2  927.59   607.6  921.88   688.6  884.45   779.7  838.71
   930.1  754.41     960  741.06     985  737.36    1000  737.01    1015  737.45
  1119.8  744.13  1209.7  764.82  1249.7  771.25  1309.6  776.57  1410.3  781.78
  1460.6  778.46    1511  770.79  1541.2  771.48  1601.6  788.99  1662.1  799.91
  1752.7  830.48  1843.3  855.24  2115.2  906.09  2205.9  912.31  2286.4  934.74
#Mann= 3 , 0 , 0
       0      .1       0     985    .045       0    1015      .1       0
Bank Sta=985,1015
XS Rating Curve= 0 ,0
Exp/Cntr=0.3,0.1

Type RM Length L Ch R = 1 ,33361   ,975.5,973.2,973.5
XS GIS Cut Line= 4
     1607483.779      374813.939     1607850.196      375240.006
     1608088.793      375529.731     1608301.826      376356.299
#Sta/Elev= 30
      10  994.18   220.8  934.61   260.9  921.38     291  916.99   431.5  852.47
   511.8  826.28   602.5  790.12   643.1  771.13   724.3  749.63   810.7  736.82
   825.7  735.59   840.7  737.68     846  739.19   896.7   767.2   937.3  777.09
   977.9   801.8  1059.2  846.52  1160.8  898.25  1181.2  904.19  1211.6  904.63
    1232  912.01  1262.5  929.62  1364.1  994.97  1414.9 1025.56    1486 1058.53
  1526.7 1073.46  1557.1 1082.29  1689.2  1101.5  1719.7 1103.35  1790.9 1099.19
#Mann= 3 , 0 , 0
       0      .1       0   810.7    .045       0   840.7      .1       0
Bank Sta=810.7,840.7
XS Rating Curve= 0 ,0
Exp/Cntr=0.3,0.1

Type RM Length L Ch R = 1 ,32387.8 ,679.7,670.9,660.7
XS GIS Cut Line= 3
     1606691.295       375009.93     1607098.452      375515.037
     1607739.418      376390.385
#Sta/Elev= 30
    10.1  981.53      71  959.69   141.9  931.24   202.7  911.15     223  907.78
   283.8  908.85   314.3  901.38   375.1  875.54   415.6  855.99   506.9  803.48
   608.2  741.87   633.8  735.31   648.8  734.24   663.8  735.13   699.5  738.48
   902.3  746.08     953   765.5  1003.7  780.48  1054.4  799.45  1115.2  818.81
  1155.8  829.13  1196.3  836.45  1216.6  838.03  1277.4  834.64  1328.1   836.9
  1449.8  856.17  1581.6  884.53  1652.6  873.69  1672.9  873.12  1733.7   888.3
#Mann= 3 , 0 , 0
       0      .1       0   633.8    .045       0   663.8      .1       0
Bank Sta=633.8,663.8
XS Rating Curve= 0 ,0
Exp/Cntr=0.3,0.1

Type RM Length L Ch R = 1 ,31716.9 ,106.2,106.7,107.1
XS GIS Cut Line= 4
     1606035.153      375538.252     1606640.167      375989.882
     1607100.319      376305.171     1607739.418      376697.152
#Sta/Elev= 30
    10.1  967.93   191.3  937.25   231.5   927.5   271.8  912.37     302  912.74
   422.8  903.22     453  897.85   513.4  880.68   553.7   862.1   674.5  815.69
   744.9  786.76   815.8  763.32   886.8  746.76   973.3  733.08   988.3  732.22
  1003.3  734.56  1018.7  742.27  1049.1  766.17  1069.4  779.28  1089.7  786.68
  1160.7  821.59  1191.1  834.37  1312.8   861.8  1383.7  881.58  1566.1  937.01
  1748.5  997.53  1768.7 1001.38    1789 1001.42  1981.5  991.64  2062.5  985.15
#Mann= 3 , 0 , 0
       0      .1       0   973.3    .045       0  1003.3      .1       0
Bank Sta=973.3,1003.3
XS Rating Curve= 0 ,0
Exp/Cntr=0.3,0.1

Type RM Length L Ch R = 1 ,31610.2 ,274.9,254.6,234.6
XS GIS Cut Line= 4
     1606014.626      375708.349     1606677.784       376140.63
     1606898.837      376297.823     1607709.364      376749.753
#Sta/Elev= 30
    10.1  894.87    50.7  897.21    81.2   895.1     203  878.95   324.8  858.22
   365.4  848.09     477  811.67   558.2  779.26   598.8  767.16   690.1   750.2
   801.7  744.07   877.1  732.33   892.1  731.93   907.1  733.73   922.2  739.79
   972.4  770.77   992.5  778.94  1042.8  784.77  1143.6  800.99  1204.1  813.96
  1284.8  835.72  1486.5  898.19  1587.4  933.41  1647.9  956.86  1688.3  975.11
  1748.8 1009.01    1779 1021.85  1799.2 1024.58  1879.9 1022.57  1990.9 1011.03
#Mann= 3 , 0 , 0
    10.1      .1       0   877.1    .045       0   907.1      .1       0
#XS Ineff= 2 , 0
          824.54  771.24
Permanent Ineff=
       F       F
Bank Sta=877.1,907.1
XS Rating Curve= 0 ,0
Exp/Cntr=0.3,0.1

Type RM Length L Ch R = 1 ,31355.5 ,424.5,419.9,415.3
XS GIS Cut Line= 4
     1605823.047      376125.893     1606569.714      376440.279
      1606839.89      376425.542     1607709.364      376793.963
#Sta/Elev= 30
    10.1  869.48    50.6  852.39   121.5  834.72   232.9  795.54   364.6   819.7
   415.2  826.29   486.1  826.29   567.1  831.99   587.4  830.75   688.6  796.41
   779.8  774.33   810.2  768.99   905.4  733.92   920.4  731.71   935.4  732.81
  1010.6  741.25  1141.7  748.63    1162  752.77  1202.6  766.44  1334.6  795.01
  1395.5  823.66  1517.3  869.72  1659.5  930.72  1700.1  951.49  1740.7  983.14
  1771.2 1001.21  1862.6 1044.41  1882.9    1047  1903.2 1045.57    2025 1024.97
#Mann= 3 , 0 , 0
       0      .1       0   905.4    .045       0   935.4      .1       0
Bank Sta=905.4,935.4
XS Rating Curve= 0 ,0
Exp/Cntr=0.3,0.1

Type RM Length L Ch R = 1 ,30935.6 ,886.5,899.9,914.6
XS GIS Cut Line= 4
     1605413.096      376526.726     1606691.295      376790.887
     1607202.575       376680.11     1607952.452      377038.005
#Sta/Elev= 30
    10.1 1000.94   111.3  990.18   273.2   990.6   374.4  981.79   495.8  978.93
     688  960.51   738.6  953.45   920.7  911.54   991.6  904.35  1042.1  889.53
  1082.6  888.39  1092.7  885.67  1234.4  808.12  1295.1  778.69  1405.8  751.74
  1496.4  733.88  1541.7  728.08  1556.7  727.87  1571.7  728.78  1586.9  732.83
  1717.7  789.08  1858.8  862.35  1960.1  901.58  2041.1  944.15  2101.9  985.21
    2183 1024.62  2274.2  1063.8  2314.7 1071.48  2547.8 1046.07  2659.3 1055.19
#Mann= 3 , 0 , 0
       0      .1       0  1541.7    .045       0  1571.7      .1       0
Bank Sta=1541.7,1571.7
XS Rating Curve= 0 ,0
Exp/Cntr=0.3,0.1

Type RM Length L Ch R = 1 ,30035.7 ,534.9,546,555.7
XS GIS Cut Line= 3
     1606197.058      377447.029     1606963.978      377625.977
     1607782.025       377898.66
#Sta/Elev= 30
    10.1  955.25   111.1   912.8   151.4  903.08   171.6   896.3   181.7  894.71
   232.2  894.71   262.5  898.17   323.1  883.58   363.5  880.06   403.9   862.4
     525  797.03   545.2   788.9   575.5   779.7   595.7  766.01     626  740.75
   636.1  735.51   716.8  727.38   752.3  726.26   767.3  725.92   782.3  726.98
   970.1  753.99  1010.7  770.34    1102  800.37  1183.2  813.29  1233.9  818.09
  1294.8  827.95  1325.2  835.23  1396.2  845.71  1538.2  876.16  1649.8  905.25
#Mann= 3 , 0 , 0
       0      .1       0   752.3    .045       0   782.3      .1       0
Bank Sta=752.3,782.3
XS Rating Curve= 0 ,0
Exp/Cntr=0.3,0.1

Type RM Length L Ch R = 1 ,29489.7 ,1185,1152.1,1119.1
XS GIS Cut Line= 3
     1606316.357       377839.01     1606760.301      378140.771
      1607364.48      378588.887
#Sta/Elev= 30
    10.1  868.29    30.4  858.48    91.2  832.76   192.4  794.99   243.1  781.71
   324.1  765.09   334.2  759.89   364.6  734.77   374.7  730.13   384.9  728.78
   425.4  728.59   455.8  731.46   491.4  725.42   506.4  723.57   521.4  725.06
   546.8  728.74   576.9  730.19   586.9  732.93     607  743.94     617  747.47
   637.1  751.06   707.3  778.54   737.4  791.65   797.6  821.17   917.9  869.28
   998.2  894.21  1148.6  946.99  1238.9  968.61  1258.9  975.66    1289  988.59
#Mann= 3 , 0 , 0
    10.1      .1       0   491.4    .045       0   521.4      .1       0
#XS Ineff= 2 , 0
          459.15  766.19  564.38          771.02
Permanent Ineff=
       F       F
Bank Sta=491.4,521.4
XS Rating Curve= 0 ,0
Exp/Cntr=0.3,0.1

Type RM Length L Ch R = 1 ,28337.6 ,839.2,849.7,859.5
XS GIS Cut Line= 3
     1605609.087      379458.062     1606435.656      379023.475
     1607091.798      378665.579
#Sta/Elev= 30
    10.2  993.62    40.6  990.18   121.8  964.85     203  943.92   274.1  931.58
   345.1  925.85   385.7  918.28   436.5  886.47   497.4  872.19   558.3  851.82
   588.7  832.47   669.9  790.06     812  725.19   939.1  721.84   954.1  719.99
   969.1  721.36   994.5  728.87  1075.3   772.8  1135.9  790.05  1186.4  816.32
  1226.8  832.57  1287.4  853.47  1398.5  886.14    1449   904.6  1489.4  924.08
  1539.9  961.18  1570.2  977.97  1590.4  983.27  1640.9  982.27  1681.3  988.19
#Mann= 3 , 0 , 0
       0      .1       0   939.1    .045       0   969.1      .1       0
Bank Sta=939.1,969.1
XS Rating Curve= 0 ,0
Exp/Cntr=0.3,0.1

Type RM Length L Ch R = 1 ,27487.9 ,595.8,592.9,590.8
XS GIS Cut Line= 3
     1606009.589         379833.     1606887.286      379705.181
     1607637.162      379568.839
#Sta/Elev= 30
    10.1 1075.28    60.5 1058.37   120.9 1030.18   141.1 1018.26   201.6  977.26
   292.3  919.06   362.8  875.98   413.2  854.61   493.9  827.06   544.3   806.2
   594.7  782.86   695.5  729.35   705.5  725.34   715.6  723.68   882.1  720.45
   897.1  719.69   912.1  720.15   927.6  724.02   937.8  730.15   988.6  768.53
   998.7  774.98  1008.9  778.36  1029.2  782.53  1039.4  787.06    1141  836.82
    1263  889.29  1374.7  942.29  1476.4  981.06    1578  1024.5  1649.1 1051.79
#Mann= 3 , 0 , 0
       0      .1       0   882.1    .045       0   912.1      .1       0
Bank Sta=882.1,912.1
XS Rating Curve= 0 ,0
Exp/Cntr=0.3,0.1

Type RM Length L Ch R = 1 ,26895   ,782.5,809.8,836.5
XS GIS Cut Line= 3
     1606248.186        380472.1     1607185.532      380233.503
     1608284.783      379926.735
#Sta/Elev= 30
    10.1  941.72   110.8  909.58   151.1   887.9   191.4  862.58   211.6     853
     403  785.31   493.7  761.95   604.5  729.42   654.9  719.02   710.4  715.64
   725.4  714.83   740.4  715.14   856.4  722.56   916.9  756.36   947.1  764.82
   987.4  787.21  1078.3  832.27  1118.7   851.1  1179.3  874.94  1310.6  951.12
  1411.6  989.19  1532.8  1008.7  1593.4 1012.03  1623.7 1018.71  1674.2 1020.54
  1916.6  1042.5  1967.1 1039.11  2027.7 1041.42    2058 1051.06  2108.5  1073.6
#Mann= 3 , 0 , 0
       0      .1       0   710.4    .045       0   740.4      .1       0
Bank Sta=710.4,740.4
XS Rating Curve= 0 ,0
Exp/Cntr=0.3,0.1

Type RM Length L Ch R = 1 ,26085.2 ,824.2,826.5,829.4
XS GIS Cut Line= 4
     1606507.959      380531.133     1606929.892      380821.474
      1607364.48      381128.242     1608361.475      381494.659
#Sta/Elev= 30
      10  870.37    60.3  869.02   150.6  848.12   180.8  837.85   271.2  797.26
   331.4  781.42   391.7  771.12   502.1  742.57   682.8  718.49   858.5  713.06
   873.5  712.43   888.5  713.35   933.7  716.88   943.8  720.24   953.8  725.71
   983.9  749.03    1014  760.93  1054.2  782.15  1155.4  825.25  1246.5  856.18
  1327.4  886.45  1408.3   920.8  1539.8  983.47  1651.1 1020.78    1732 1053.44
  1782.6 1065.45    1813 1070.42  2005.2 1075.23  2065.9 1080.58  2106.3  1087.4
#Mann= 3 , 0 , 0
       0      .1       0   858.5    .045       0   888.5      .1       0
Bank Sta=858.5,888.5
XS Rating Curve= 0 ,0
Exp/Cntr=0.3,0.1

Type RM Length L Ch R = 1 ,25258.7 ,721.4,691,660.6
XS GIS Cut Line= 4
     1605890.291      380582.877     1606290.793      380829.996
     1606844.679       381307.19     1607586.035      381605.436
#Sta/Elev= 30
      10 1082.14      30  1077.5    50.1 1070.32   260.3  965.37   310.4  937.74
   440.6   859.9   572.1  793.65   673.7  750.43   780.5  711.44   795.5  710.13
   810.5  710.37     958  718.17   988.5  727.54   998.6  732.41  1029.1  752.64
  1049.4  758.28  1059.5  763.26  1140.8  809.28  1201.7  835.37  1221.9  839.95
  1242.2  842.13  1302.9  839.69  1353.4   842.1  1454.6  857.75  1484.9  865.55
  1515.3  876.78  1596.2   892.6  1768.2  935.22  1940.1  987.52  2000.8 1009.15
#Mann= 3 , 0 , 0
       0      .1       0   780.5    .045       0   810.5      .1       0
Bank Sta=780.5,810.5
XS Rating Curve= 0 ,0
Exp/Cntr=0.3,0.1

Type RM Length L Ch R = 1 ,24567.7 ,992.9,979.9,963.7
XS GIS Cut Line= 4
     1605208.584       381946.29     1606094.802       381758.82
     1606827.636       381562.83     1607560.471      381716.214
#Sta/Elev= 30
    10.1 1033.24   171.1 1013.18   382.5  1053.4   432.8 1052.54   452.9 1049.07
   553.6 1016.71   634.1   981.2   714.6   935.4     775  890.22   805.2  871.42
   875.6  837.41   946.3  811.29    1007  771.37  1047.4  753.82  1077.8   729.8
  1087.9  724.35  1143.7  709.93  1158.7  709.18  1173.7  709.89  1300.3     726
  1350.9  735.02  1421.7  761.56  1472.2  791.88  1674.5  879.22  1806.1  925.96
  1917.4  960.13  2018.5   978.9  2220.9  994.53  2291.7  997.58  2413.1  991.49
#Mann= 3 , 0 , 0
       0     .08       0  1143.7    .045       0  1173.7     .08       0
Bank Sta=1143.7,1173.7
XS Rating Curve= 0 ,0
Exp/Cntr=0.3,0.1

Type RM Length L Ch R = 1 ,23587.8 ,869,872.7,879.8
XS GIS Cut Line= 3
     1606452.698      382772.858     1607066.836      382252.595
     1607378.627      381923.664
#Sta/Elev= 30
    10.1 1005.06    50.3  998.43   100.6  979.62   231.4  898.18   251.5  887.03
   462.8  806.19   583.5  746.53   603.7  734.93   623.8  721.01   633.8  716.76
   643.9  714.94   779.8  707.94   794.8  707.12   809.8  708.26     815  709.31
   855.2  727.86   885.5  743.51   905.6  747.88   925.7  754.93   935.8  761.45
   976.1  801.49   986.2  808.27   996.2  812.74  1006.3  814.07  1036.5   813.5
    1097  830.37  1137.2   835.6  1187.6  845.77  1207.7  852.32  1258.1  880.62
#Mann= 3 , 0 , 0
       0     .08       0   779.8    .045       0   809.8     .08       0
Bank Sta=779.8,809.8
XS Rating Curve= 0 ,0
Exp/Cntr=0.3,0.1

Type RM Length L Ch R = 1 ,22715.1 ,535.2,538.3,541.1
XS GIS Cut Line= 3
     1606623.125      383326.744     1607262.224      383122.232
     1607778.806      382787.984
#Sta/Elev= 30
      10  999.45    40.1 1000.09    60.1  998.02   150.2  981.19   170.3   975.3
   190.3  966.57   230.4  941.45   240.4  936.49   320.5  903.16   470.7  845.95
   560.9  808.46   610.9  785.53   751.7   716.5   777.1  706.22     782  704.41
   792.1  702.62   802.2  703.52   807.1  704.76   822.3  707.77   923.2  710.12
   933.3  711.03   943.4  713.91   953.5  719.51   983.7  739.37   993.8  744.27
  1003.9  747.53    1014  752.12  1054.3  774.33    1135   817.3  1286.3  888.89
#Mann= 3 , 0 , 0
       0      .1       0   777.1    .045       0   807.1      .1       0
Bank Sta=777.1,807.1
XS Rating Curve= 0 ,0
Exp/Cntr=0.3,0.1

Type RM Length L Ch R = 1 ,22176.8 ,325.7,347.5,369.5
XS GIS Cut Line= 5
     1606691.295      383531.256     1607577.513      383497.171
     1608003.579      383258.574      1608455.21      381792.906
      1608523.38      381622.479
#Sta/Elev= 30
    10.1  950.07   221.7   994.2   332.6   974.7     383  956.26   574.5  864.58
   876.8  760.79   926.7  735.85   986.5  712.11  1006.5  707.63  1101.1  702.92
  1116.1  700.23  1131.1  701.46  1175.9  711.54  1215.7  730.83  1235.7  736.25
  1375.2  735.39  1415.8  748.15  1629.1  834.35  1690.1  848.69    1883  859.87
  1933.8  856.25  2045.5  837.29  2329.9   880.5    2462  873.38  2614.3  854.62
    2655  870.43  2776.8  939.59  2847.9  973.05  2966.8 1018.06  3092.4 1055.29
#Mann= 3 , 0 , 0
       0      .1       0  1101.1    .045       0  1131.1      .1       0
Bank Sta=1101.1,1131.1
XS Rating Curve= 0 ,0
Exp/Cntr=0.3,0.1

Type RM Length L Ch R = 1 ,21829.3 ,625.7,641.5,660.5
XS GIS Cut Line= 4
     1606708.338      383607.948     1607662.726      383599.427
     1608165.485      383727.247     1609682.281      384332.261
#Sta/Elev= 30
    10.2  934.23   243.7  995.27   284.3  996.66   436.6  951.53   619.4  865.91
   720.9  835.06     924  759.21   994.3  740.62  1064.2  714.27  1228.7  700.54
  1243.7  697.94  1258.7  699.59  1283.6  709.95  1323.5  740.49  1403.3  777.63
  1453.2  810.97  1615.2  871.08  1807.9  966.25  1878.9  988.11  1929.6  993.64
  2020.9  972.63    2102  944.69  2193.3  902.52  2233.9  928.53  2467.2  998.91
  2680.2  984.51  2852.6 1033.67  2933.8  1050.1  3014.9 1056.96  3106.2 1052.82
#Mann= 3 , 0 , 0
       0      .1       0  1228.7    .045       0  1258.7      .1       0
Bank Sta=1228.7,1258.7
XS Rating Curve= 0 ,0
Exp/Cntr=0.3,0.1

Type RM Length L Ch R = 1 ,21187.8 ,795.3,800,803
XS GIS Cut Line= 3
     1607164.306      383763.594     1607494.344      384091.249
     1607781.388      384442.012
#Sta/Elev= 30
    10.1  880.08   151.7  812.93     182   799.4   232.5  768.18   313.4  716.77
   323.5  711.76   333.6  709.25   424.6  704.05   450.1  699.15  454.97  697.45
   465.1  698.19   480.1  701.97   495.3  705.84   525.5   707.8   535.6  711.23
   565.8   728.6   575.9  733.21     596  737.56   606.1   740.9   616.1  745.73
   636.3  757.45   686.6  788.58   696.7  794.46   706.8  799.23   767.2  817.54
   807.5  830.76   827.7  838.15   857.9  851.33     878  858.68   918.3  868.18
#Mann= 3 , 0 , 0
    10.1      .1       0   450.1    .045       0   480.1      .1       0
Bank Sta=450.1,480.1
XS Rating Curve= 0 ,0
Exp/Cntr=0.3,0.1

Type RM Length L Ch R = 1 ,20387.8 ,871.5,872,871.1
XS GIS Cut Line= 3
     1606573.667       384145.97     1606847.624      384519.512
     1607142.926      384962.839
#Sta/Elev= 30
    10.1  848.28    30.2  838.97    70.5  824.89   110.8  814.96   181.3  795.95
   201.4  789.52   211.5  784.63   271.9  749.43     292  740.06   322.2  729.09
   362.5  716.49   382.7  711.14   402.8  707.81     433  704.79   448.2  700.43
  463.43     697   478.2  698.81   513.5   704.3   583.8   707.5   593.9  708.58
   644.1  723.83   654.2  729.26   714.5  768.48   744.6  786.26   764.7  794.26
   794.9  803.23   825.1  813.34   885.4  835.17   935.6  857.77   995.9  888.58
#Mann= 3 , 0 , 0
    10.1      .1       0   448.2    .045       0   478.2      .1       0
Bank Sta=448.2,478.2
XS Rating Curve= 0 ,0
Exp/Cntr=0.3,0.1

Type RM Length L Ch R = 1 ,19515.8 ,668.8,654.7,640.6
XS GIS Cut Line= 3
     1605788.035       384195.92     1606231.144      384835.019
     1606725.381      385422.991
#Sta/Elev= 30
    10.1     900   111.1  845.23   161.6  820.04     202  807.05   272.7  794.16
   292.9  789.19     303  784.21   313.1  777.17   363.6  738.54     404  711.09
   424.2  701.49   449.6  697.57  464.62  695.86   479.6  698.03   515.1   700.8
   656.5  706.41   676.7  709.66     707   723.5   727.2  729.36   828.2  788.88
   939.4  831.72  1030.3  871.77  1171.8  949.51  1232.5  979.63  1242.6   980.6
  1252.7  979.72  1333.5   966.8  1454.8  953.99  1495.3  951.69  1545.8   951.4
#Mann= 3 , 0 , 0
    10.1      .1       0   449.6    .045       0   479.6      .1       0
Bank Sta=449.6,479.6
XS Rating Curve= 0 ,0
Exp/Cntr=0.3,0.1

Type RM Length L Ch R = 1 ,18861.1 ,885.4,873.3,864.5
XS GIS Cut Line= 3
     1605203.125       384814.82     1605604.313      385029.259
     1606006.996      385242.179
#Sta/Elev= 30
    10.1  769.78    80.9   760.9   131.4  753.14   161.7  747.34   222.4  734.55
   262.8  726.59   283.1  723.03   333.6  715.44   363.9  708.48   394.2  702.87
   414.5  697.55   419.7  696.54   424.6  695.59   434.7  695.21   449.7  696.84
     465  698.71   495.4  701.02   657.4  710.19   667.5  710.99   677.6  712.71
   687.7  715.46   718.1  725.33   728.2  728.15   748.5  731.65   758.6  735.65
   819.3  765.45   829.4  770.13   839.6  774.24   869.9  784.57   910.4   796.4
#Mann= 3 , 0 , 0
       0      .1       0   419.7    .045       0   449.7      .1       0
Bank Sta=419.7,449.7
XS Rating Curve= 0 ,0
Exp/Cntr=0.3,0.1

Type RM Length L Ch R = 1 ,17987.8 ,805.3,800,791.1
XS GIS Cut Line= 3
     1604867.731       385806.45     1605330.922      385847.351
     1605779.223      385936.311
#Sta/Elev= 30
    10.1  872.76    50.5  857.74    60.7  853.58      91  840.04   101.1  835.94
   161.7  813.45     182  806.55   212.3  797.17   242.6  788.35   252.7  784.63
   262.8   780.3   293.1  765.21   333.6  746.49   394.2  715.61   414.4  705.71
   424.6  701.39   434.7  698.15     450     695   454.9   694.2     465  693.55
     480  694.15   536.1  698.92   627.5  702.11   637.7  703.48   647.8  706.66
   698.6  727.35   708.7  729.88   718.9  731.55   729.1  734.52     922  817.48
#Mann= 3 , 0 , 0
       0      .1       0     450    .045       0     480      .1       0
Bank Sta=450,480
XS Rating Curve= 0 ,0
Exp/Cntr=0.3,0.1

Type RM Length L Ch R = 1 ,17187.8 ,554.9,569,583.4
XS GIS Cut Line= 3
     1604914.745      386682.717     1605367.655      386642.417
     1605822.099      386597.027
#Sta/Elev= 30
    10.1  789.72    30.3  787.54    60.6  782.83    70.7  782.51   111.1  790.19
   131.4  791.74   151.6  791.01   252.6  771.89   262.7  769.59   272.8  765.97
   313.2   745.8   363.8  725.85   414.3  702.86   424.4  699.17   439.7  695.32
   454.7  693.32   469.7  693.95   505.4  696.21   606.9  696.51   667.8  698.25
     678  698.96   688.1  701.65   698.3  706.71   718.6  717.94   728.7  721.48
   738.9  723.68     749  727.25   759.2  732.58   840.4  778.67   911.4  819.72
#Mann= 3 , 0 , 0
       0      .1       0   439.7    .045       0   469.7      .1       0
Bank Sta=439.7,469.7
XS Rating Curve= 0 ,0
Exp/Cntr=0.3,0.1

Type RM Length L Ch R = 1 ,16618.8 ,862.4,876.9,891.4
XS GIS Cut Line= 4
     1604782.518      387033.521     1605285.276      387067.607
     1605779.513      387263.597     1606299.314      387434.024
#Sta/Elev= 30
    10.1   916.9    90.7  900.05   231.8  864.61   282.2  850.43   322.5  835.73
   372.9  811.87   403.1  789.05   433.4  769.66   463.6  742.27   493.8  726.43
     524  705.66     534  702.14   744.7  696.23   754.7  695.47   769.8  691.94
   784.8  689.58   799.8  691.16   814.9  694.82     845  706.42     855  708.81
   875.1  710.91   955.3  725.97  1035.6  745.21    1147  784.58  1177.4  798.08
  1369.9  863.66  1461.1  901.96  1521.8  930.54  1542.1  938.26  1582.6  950.68
#Mann= 3 , 0 , 0
       0      .1       0   769.8    .045       0   799.8      .1       0
Bank Sta=769.8,799.8
XS Rating Curve= 0 ,0
Exp/Cntr=0.3,0.1

Type RM Length L Ch R = 1 ,15742   ,823.4,812.1,800.8
XS GIS Cut Line= 3
     1604220.111      386956.829     1604791.039      387570.365
     1605242.017      388082.014
#Sta/Elev= 30
    10.1  938.37     101  907.34   181.8   878.8   222.1  865.49   262.5  853.28
   323.1  837.62   373.6  822.79   454.4   803.9   525.1   790.8   636.1  764.18
   656.3  760.43   716.9  751.57   817.9  732.08   908.3  710.24   958.4   699.4
  1003.6  687.45  1018.6  686.29  1033.6  689.17  1048.7  692.12  1058.7  692.64
    1159  694.19  1169.1  695.45  1179.1  698.35  1199.2  706.05  1219.2  709.72
  1259.3  731.44  1359.6  780.32  1379.7  789.63  1419.8  805.85  1520.1  854.01
#Mann= 3 , 0 , 0
       0      .1       0  1003.6    .045       0  1033.6      .1       0
Bank Sta=1003.6,1033.6
XS Rating Curve= 0 ,0
Exp/Cntr=0.3,0.1

Type RM Length L Ch R = 1 ,14929.9 ,817.1,850.9,884.8
XS GIS Cut Line= 4
     1603325.371      387672.621     1604177.504        388183.9
     1604722.869      388465.104     1606410.091      388499.189
#Sta/Elev= 30
    10.1 1072.28    91.3 1079.58   192.7 1056.78   344.8 1015.08   476.6 1014.91
   537.4 1001.61   638.8   963.3   730.1  915.39   892.3  842.96  1094.3  740.88
  1240.3   687.2  1255.3  685.78  1270.3  686.15  1486.6  697.19  1678.1  776.64
  1738.7  793.01    2153  846.92  2274.3  867.51  2506.7  868.26  2567.3  876.79
  2638.1  893.84  2688.6  892.67    2729   899.1  2769.4  911.41  2880.6  959.41
  3032.2   997.5  3173.6 1052.59    3204 1071.36  3264.6 1083.79  3294.9 1096.61
#Mann= 3 , 0 , 0
       0      .1       0  1240.3    .045       0  1270.3      .1       0
Bank Sta=1240.3,1270.3
XS Rating Curve= 0 ,0
Exp/Cntr=0.3,0.1

Type RM Length L Ch R = 1 ,14078.9 ,833.1,822.9,812.7
XS GIS Cut Line= 4
     1603427.627      387894.175     1603990.035      388703.701
     1603972.992      389163.853     1603734.395      390552.829
#Sta/Elev= 30
    10.2 1084.92   111.8 1074.67   193.1 1042.18   304.9 1009.48   416.6  956.87
   518.3  923.28     630  874.36   782.5  816.04   945.1  760.45  1075.8  697.57
    1236  691.59    1261  687.04    1276   685.2    1291  686.52  1336.1  697.11
  1346.1  704.16  1376.1  735.76  1416.2  765.21  1659.1  899.77  1750.4  960.77
  1770.6  971.01  1811.2  983.41    1872  991.82  1912.6 1001.16  2054.5  1012.4
  2247.2 1047.43  2490.5 1065.33  2713.6 1056.35  2774.4 1059.39  2855.5 1068.85
#Mann= 3 , 0 , 0
       0      .1       0    1261    .045       0    1291      .1       0
Bank Sta=1261,1291
XS Rating Curve= 0 ,0
Exp/Cntr=0.3,0.1

Type RM Length L Ch R = 1 ,13256   ,794.7,791.3,787.9
XS GIS Cut Line= 4
     1603103.817       387860.09     1603112.338      388720.744
     1603274.243      389240.545     1603521.362      389589.919
#Sta/Elev= 30
    10.1 1059.17   141.8 1015.13     162 1009.95   263.3 1002.77   384.8   989.3
   415.2  984.89   435.4  978.67   496.2  950.65   607.6   893.4   698.7   848.8
   810.1  789.36   860.7  759.91   931.3  722.51   961.5  709.13  1027.2  685.88
  1042.2  682.79  1057.2  683.39  1092.6  686.63  1253.9  692.86  1294.2  701.49
  1324.5  719.93    1425     774  1494.7  813.61  1574.3  842.95    1634  869.32
  1713.6  900.38  1763.4  923.66  1803.2  948.59  1813.2  952.68  1833.1  958.51
#Mann= 3 , 0 , 0
       0      .1       0  1027.2    .045       0  1057.2      .1       0
Bank Sta=1027.2,1057.2
XS Rating Curve= 0 ,0
Exp/Cntr=0.3,0.1

Type RM Length L Ch R = 1 ,12464.7 ,863.5,876.9,890.6
XS GIS Cut Line= 4
     1602081.258      388490.668     1602430.632      389138.289
     1602631.942      389577.032     1602745.921      389973.379
#Sta/Elev= 30
    10.1  967.33    60.5  958.37   181.4  950.41   262.1  930.57   342.7  907.72
     383  900.13   423.4  879.54   453.6  867.17   584.6  827.01   614.9  814.95
   675.4  783.85   836.4  693.33   846.5  690.15   901.9  682.31   916.9  681.49
   931.9  684.19   957.1  688.33  1077.8   690.8    1118  701.67  1178.3  740.58
  1228.6  770.47    1289  798.08  1369.5  827.98  1449.9  862.16  1480.1  872.72
  1510.3  881.01  1550.5  883.18  1570.6  887.04  1610.9  903.33    1631  907.91
#Mann= 3 , 0 , 0
       0      .1       0   901.9    .045       0   931.9      .1       0
Bank Sta=901.9,931.9
XS Rating Curve= 0 ,0
Exp/Cntr=0.3,0.1

Type RM Length L Ch R = 1 ,11587.8 ,708,704.6,701
XS GIS Cut Line= 3
      1601713.23      388993.384     1601697.665      389448.116
      1601680.18      389902.785
#Sta/Elev= 30
    10.1  768.07    50.6  756.23    60.7  754.23    80.9   751.7   101.1  747.32
     182  725.01   242.7  705.88   252.8  703.41     273  700.58   414.6  685.74
     440  680.88   444.9  679.88     455  679.34     470  681.71   485.3  684.73
   525.8  688.46   566.2  695.65   616.8  702.35   657.2   700.1   697.7  700.98
   748.2  704.24   768.4  703.51   788.7  701.47   798.8  701.14   808.9  701.96
     819  704.17   829.1  707.66   849.3   716.4   889.8  738.33     910  748.18
#Mann= 3 , 0 , 0
       0      .1       0     440    .045       0     470      .1       0
Bank Sta=440,470
XS Rating Curve= 0 ,0
Exp/Cntr=0.3,0.1

Type RM Length L Ch R = 1 ,10883.2 ,909.8,895.4,883.1
XS GIS Cut Line= 4
     1601246.168      388499.189     1600990.528      389308.715
     1601034.751      389789.759     1601280.253      390322.753
#Sta/Elev= 30
    10.1  982.69    40.4  971.28   151.6  934.95   212.2  918.55     283  903.74
   424.5  882.98   596.3   841.4   687.2  830.23   707.4  825.13   818.6  783.01
     859  758.13   929.4  709.43   979.8  681.34   989.8  679.19  1025.1  678.52
  1040.1  677.46  1055.1  678.48  1090.5  684.52  1191.1  687.74  1221.3  692.41
  1271.6   708.2  1301.8   714.1  1311.9  718.32  1463.5  794.99  1483.8  802.57
  1777.2  890.26  1797.4  894.09  1858.1  900.54  1898.6  908.05  1918.8  908.55
#Mann= 3 , 0 , 0
       0      .1       0  1025.1    .045       0  1055.1      .1       0
Bank Sta=1025.1,1055.1
XS Rating Curve= 0 ,0
Exp/Cntr=0.3,0.1
